HEC-RAS study LYNNCMPRN.prj: LYNNCMPRN

--- LYNNCMPRN.g01 (geometry) --- (continued)

Type RM Length L Ch R = 1 ,4076    ,25.4,25.6,27.3
XS GIS Cut Line= 3
2152917.92881824 648744.515993262152998.66042475648871.325544988
2153015.79685066648882.369019463
#Sta/Elev= 30
       0 1570.78     5.5  1570.8      15 1571.41    19.1 1571.19    19.8 1571.07
    24.5 1569.59    29.2 1568.38      34 1567.84    42.7 1566.08    48.9 1563.97
    57.7 1561.91    63.8 1560.14    67.2  1559.3    71.6 1558.63    74.5 1558.45
    86.1 1557.91    95.6 1557.75   105.1 1557.28   108.5 1557.22   109.8 1557.23
   112.2  1557.8   114.6 1558.57   119.3 1560.54   124.1 1561.87   133.6 1563.84
     143 1566.15   158.6 1569.59   161.4 1570.14   168.5 1571.23   170.7  1571.7
#Mann= 5 ,-1,0
       0     .06       0      50      .1       0    95.6    .045       0
   112.2      .1       0     140     .06       0
Bank Sta=95.6,112.2
XS Rating Curve= 0 ,0
Exp/Cntr(USF)=0,0
Exp/Cntr=0.3,0.1

Type RM Length L Ch R = 1 ,4050    ,29.7,29,28.4
XS GIS Cut Line= 4
 2152831.3672385648747.987708265 2152883.8833978648784.642963101
2152935.97543392648819.6138404952152988.49461418648902.455024049
#Sta/Elev= 30
       0 1565.86      44 1565.89    61.8 1566.06    76.2 1566.44    84.8 1566.34
    96.3 1565.79   107.9 1564.62   117.4 1564.29   126.8 1562.91   134.6 1562.93
   138.1 1562.48   142.6 1561.47   145.5 1560.15   149.6  1557.8   152.61556.827
     157 1556.16     172 1556.37   174.4 1556.79     176 1557.16   177.3    1558
   180.2  1559.5   183.1  1560.7   186.9 1561.78   194.9 1564.38   197.6 1565.03
   199.7 1565.46   213.9 1566.61   218.6 1567.21   223.4 1568.05   224.9 1568.59
#Mann= 4 ,-1,0
       0      .1       0   152.6    .045       0   174.4      .1       0
  196.79     .06       0
Bank Sta=152.6,174.4
XS Rating Curve= 0 ,0
Exp/Cntr(USF)=0,0
Exp/Cntr=0.3,0.1

Type RM Length L Ch R = 1 ,4021    ,17.6,24.6,31.8
XS GIS Cut Line= 3
2152811.47702276648765.308211851 2152903.2944159648824.545239682
   2152966.76266648915.516389565
#Sta/Elev= 30
       0 1565.43    21.9 1566.07    34.2 1565.88    43.7 1565.25    51.4 1565.76
    61.2 1565.44    73.5 1566.46    86.5 1565.08    95.7 1565.17   104.6 1563.65
     110 1563.68   114.9 1562.97   119.8  1561.5   124.7 1559.45   127.6 1558.68
   130.5 1558.09   139.1 1557.25   144.2 1555.29   149.1 1554.29   163.7 1555.19
   168.6 1556.83   173.4 1560.38   178.3 1563.07   180.7 1563.87   183.2 1564.27
     193  1564.6   207.6 1565.69   212.5 1566.71   215.7  1567.8   220.2 1570.24
#Mann= 4 ,-1,0
       0      .1       0   144.2    .045       0   163.7      .1       0
  179.27     .06       0
Bank Sta=144.2,163.7
XS Rating Curve= 0 ,0
Exp/Cntr(USF)=0,0
Exp/Cntr=0.3,0.1

Type RM Length L Ch R = 1 ,3997    ,56.3,51.4,48.5
XS GIS Cut Line= 4
2152815.69077611648777.9502099062152900.06726645648828.670909155
2152907.65167008648887.924062483 2152929.4568305648916.839601307
#Sta/Elev= 30
       0 1565.13      14 1565.29    29.6 1564.93    40.6 1565.06    45.1 1564.68
    51.9 1563.39    61.2  1563.9    65.9 1563.92    83.9  1562.7    93.9 1561.25
    98.4 1561.26     103 1558.82     107 1556.45   111.1 1554.34   119.1 1551.02
     122 1550.28   123.2 1550.01   127.2 1550.58   131.2 1551.48   138.51552.106
   155.4 1552.53   159.1 1553.35   159.8 1553.59     168 1558.72   170.9 1560.08
   174.8 1561.56     179 1562.71   184.8 1564.61   190.9 1567.15   194.4 1567.98
#Mann= 4 ,-1,0
       0      .1       0     122    .045       0   138.5      .1       0
  148.45     .06       0
Bank Sta=122,138.5
XS Rating Curve= 0 ,0
Exp/Cntr(USF)=0,0
Exp/Cntr=0.3,0.1

Type RM Length L Ch R = 1 ,3945    ,63.6,67.4,68.2
XS GIS Cut Line= 4
2152846.71744835648808.1111738572152841.00530639 648826.39002816
2152872.23168249648888.0811614332152888.98729893648926.162107898
#Sta/Elev= 30
       0 1562.39     2.9 1561.23     6.1 1559.72     9.3 1557.84    13.7 1554.45
    17.9 1550.75    18.8 1549.81    20.6 1548.93    22.3 1547.84    23.6 1547.51
    26.8 1545.72    29.5 1545.06      35 1543.04    37.81542.193    40.2  1541.6
    43.9 1541.35    52.7 1542.16    67.1 1544.05    71.6 1544.87    80.1 1547.85
      85 1548.95    89.5 1550.63    95.2 1553.06    98.2    1554   102.6 1555.01
     107 1556.84   111.3 1559.31   116.4 1561.15   128.5 1566.43   129.9 1566.71
#Mann= 4 ,-1,0
       0      .1       0    37.8    .045       0    52.7      .1       0
   79.15     .06       0
Bank Sta=37.8,52.7
XS Rating Curve= 0 ,0
Exp/Cntr(USF)=0,0
Exp/Cntr=0.3,0.1

Type RM Length L Ch R = 1 ,3878    ,71.5,84.2,92.7
XS GIS Cut Line= 3
2152799.40791299648840.9937457192152798.64629406648865.365551457
 2152823.0180998648940.004206528
#Sta/Elev= 30
       0 1545.77       1 1545.27     4.2 1543.45     8.2 1541.75    12.2  1541.2
    20.2 1541.93    24.2  1541.7    28.4 1540.97    31.8 1539.87    36.8 1538.65
    44.5 1537.62    48.51537.008    50.8 1536.68      54 1536.42    57.2 1535.98
    57.9 1535.82    62.1 1535.92    63.5 1536.97    65.4 1538.53    66.3 1539.17
    70.5  1544.5      73 1547.21    76.2 1550.39    78.9 1552.93    80.9 1554.05
    83.1 1555.39    85.7 1556.67    88.9 1558.11    99.9 1562.23   102.9  1563.1
#Mann= 4 ,-1,0
       0      .1       0   44.38     .06       0    48.5    .045       0
    63.5     .06       0
Bank Sta=48.5,63.5
XS Rating Curve= 0 ,0
Exp/Cntr(USF)=0,0
Exp/Cntr=0.3,0.1

Type RM Length L Ch R = 1 ,3794    ,51.1,45.5,40
XS GIS Cut Line= 4
2152753.79836341648829.382865142 2152748.7602542648851.275601265
2152723.24602006648891.2605950532152709.80166678648911.907584757
#Sta/Elev= 30
       0 1542.13     4.5 1540.21       8  1538.5    12.1 1536.11    16.2 1534.27
    20.3  1532.6    24.7 1531.29    35.9 1529.92    38.8  1529.4    43.7 1527.39
    47.4 1525.35    48.4 1524.82    50.3 1524.09    53.2 1523.29    56.1 1524.13
    57.9 1524.84      59 1525.43    64.8 1529.03    67.4 1530.88    70.6 1532.31
    72.2 1533.29    73.5 1533.87    75.5 1535.01    76.4 1535.39    81.7 1538.16
    82.9 1538.67    86.5 1539.73    90.2 1540.18    91.3 1539.99    94.5 1538.97
#Mann= 4 ,-1,0
       0      .1       0    47.4    .045       0      59      .1       0
   62.46     .06       0
Bank Sta=47.4,59
XS Rating Curve= 0 ,0
Exp/Cntr(USF)=0,0
Exp/Cntr=0.3,0.1

Type RM Length L Ch R = 1 ,3748    ,76.2,76.5,77.2
XS GIS Cut Line= 4
2152695.44692915648820.8108440932152689.35397771648847.848316083
2152688.97316825648901.923260063 2152692.4880396648921.569220345
#Sta/Elev= 30
       0 1536.99     9.7 1532.38    12.7 1531.04    16.4 1529.09    19.8 1527.69
      25    1526      29 1524.88      33 1524.27    34.2 1523.86    35.9 1523.03
    38.2 1522.09    39.61521.328      41 1520.58      45 1520.85    46.1 1520.99
      48 1521.39      49 1521.53      53 1521.21      57 1521.58      61 1523.99
      65 1525.89    69.9 1526.54      77 1527.74      81 1529.08    85.1  1531.1
    89.2 1533.74    94.2 1536.71    97.3 1538.33   101.4 1539.99   101.7 1540.18
#Mann= 4 ,-1,0
       0      .1       0      10     .06       0    39.6    .045       0
      48     .06       0
Bank Sta=39.6,48
XS Rating Curve= 0 ,0
Exp/Cntr(USF)=0,0
Exp/Cntr=0.3,0.1

Type RM Length L Ch R = 1 ,3672    ,54.8,55.8,56.2
XS GIS Cut Line= 4
2152631.86689735 648848.306436662152621.96585127648871.916623468
2152625.39313645648914.5672835092152632.24770681648953.409848903
#Sta/Elev= 27
       0 1521.57      .9 1521.21     5.3 1520.44     9.5 1520.01      14 1520.02
    18.3 1519.83    22.6  1518.9    30.9 1516.61    36.3 1515.26    42.31513.596
    42.9 1513.43    46.9 1513.13    50.8 1513.12      55 1513.23    56.11513.543
      59 1514.37      63 1517.57      67 1522.01      71 1527.34    75.1  1532.5
      78 1535.17    79.2 1536.19    87.3 1540.89    91.4  1543.5    95.4 1545.61
   103.5 1548.76   107.8  1550.3
#Mann= 3 ,-1,0
       0     .06       0    42.3    .045       0    56.1     .06       0
Bank Sta=42.3,56.1
XS Rating Curve= 0 ,0
Exp/Cntr(USF)=0,0
Exp/Cntr=0.3,0.1

Type RM Length L Ch R = 1 ,3616    ,50.3,52.5,53.7
XS GIS Cut Line= 3
 2152570.2280298648844.6444987342152569.58312563648869.150857278
2152569.58312563648938.155603704
#Sta/Elev= 30
       0  1526.2     6.7 1524.84    12.5 1523.39    16.5 1521.72    20.5 1519.79
    24.5 1517.41      26 1516.21    28.5 1513.99    32.5 1511.19    36.5 1510.41
    44.5 1510.28    48.5  1510.1    52.5 1509.51    56.5 1509.06    60.5 1508.95
    62.51509.497    64.5 1510.08      66 1511.28    67.1 1512.36    68.5 1513.56
    72.5  1516.8    76.5 1518.67      78  1520.2    79.1  1521.6    80.5 1523.14
      82 1525.78    84.5 1530.51      86 1532.38    88.5 1535.73    93.5  1539.2
#Mann= 4 ,-1,0
       0      .1       0   34.51     .06       0    52.5    .045       0
    62.5     .06       0
Bank Sta=52.5,62.5
XS Rating Curve= 0 ,0
Exp/Cntr(USF)=0,0
Exp/Cntr=0.3,0.1

Type RM Length L Ch R = 1 ,3563    ,72.7,77,80.1
XS GIS Cut Line= 3
2152539.27262953648856.2527738332152521.86021688648879.469324033
2152511.54175013648938.800507876
#Sta/Elev= 30
       0 1524.01     1.2 1523.78     6.2 1521.05     8.6 1520.11    11.2 1519.34
    21.2  1518.7    26.2  1517.4      29 1515.67    30.8 1514.45    38.9 1507.88
    42.9 1506.25    44.61505.994      47 1505.62    49.2 1505.53    51.1 1505.54
    52.7 1505.74    53.6 1505.97    59.2 1506.86    59.6 1506.87    63.2 1506.19
    66.5 1506.73    67.3 1506.79    71.4 1510.33    73.5  1513.8    76.9 1519.73
    79.5 1524.36    80.4 1525.68    83.5 1529.93    87.3  1533.2    89.2 1534.49
#Mann= 4 ,-1,0
       0      .1       0   29.02     .06       0    44.6    .045       0
    53.6     .06       0
Bank Sta=44.6,53.6
XS Rating Curve= 0 ,0
Exp/Cntr(USF)=0,0
Exp/Cntr=0.3,0.1

Type RM Length L Ch R = 1 ,3486    ,65.4,68.8,71.7
XS GIS Cut Line= 3
2152494.12933748648820.1381401892152465.10864973648842.709786217
2152423.83478271648923.322807743
#Sta/Elev= 30
       0 1519.31     2.5 1518.66     8.2 1516.94    13.5 1515.89    17.7 1515.32
    21.2    1515    22.7 1514.95    32.9 1515.17    36.8 1515.04    39.5 1515.06
      44 1514.59    48.2 1512.91      53 1510.17    57.1 1507.97    63.1 1505.93
      69 1503.35      71 1502.64      75 1502.42    80.9 1502.45    84.5 1502.79
    85.71503.218    93.5 1506.18    95.8 1506.73   102.5 1508.74   110.6 1512.19
   113.6  1513.6   115.9  1514.8   120.4 1517.69   124.9 1520.39   127.3 1521.51
#Mann= 3 ,-1,0
       0     .06       0      69    .045       0    85.7     .06       0
Bank Sta=69,85.7
XS Rating Curve= 0 ,0
Exp/Cntr(USF)=0,0
Exp/Cntr=0.3,0.1

Type RM Length L Ch R = 1 ,3418    ,47.4,46.5,46.1
XS GIS Cut Line= 4
2152463.17393721 648796.921589992152448.98604542 648796.92158999
 2152419.3204535648805.9502484012152363.21379052648871.730473966
#Sta/Elev= 30
       0 1520.35      11 1518.54    18.2 1518.21    27.6 1518.11    31.8 1517.53
    35.9 1515.92    37.5 1515.08    40.1 1513.43    42.5 1512.31    44.3 1511.71
      50 1510.93    52.6  1510.4    55.4 1509.42    56.2    1509    62.4 1503.91
    68.5 1501.02    72.4 1500.08    75.7 1499.56    80.9 1499.34    86.2 1499.51
    88.31500.053    89.4 1500.42    91.5 1501.54    99.4 1506.58     102 1507.82
   105.5 1508.83   117.8 1510.28   123.5 1510.42   130.2 1511.07   131.7 1511.04
#Mann= 3 ,-1,0
       0     .06       0    72.4    .045       0    88.3     .06       0
Bank Sta=72.4,88.3
XS Rating Curve= 0 ,0
Exp/Cntr(USF)=0,0
Exp/Cntr=0.3,0.1

Type RM Length L Ch R = 1 ,3371    ,78,77.7,76.1
XS GIS Cut Line= 3
2152427.56495573648772.7437814592152392.53048498648762.081116449
2152326.26963813648847.001627066
#Sta/Elev= 30
       0  1514.8     8.8 1513.49    20.3 1512.72    24.4 1511.92    28.6  1510.9
    36.6 1509.57    39.1 1509.58    47.6 1509.12    55.8  1508.3      59 1507.35
    61.9 1506.08    70.4 1501.02    73.3  1499.8    76.1 1499.01    81.8 1498.85
    85.3 1497.91    86.2 1497.64    89.2  1497.2    91.3 1497.15    95.7 1497.39
    97.61497.883   101.8 1499.49   106.5 1502.47   108.7 1503.43   110.3 1503.82
     116 1504.28   121.7  1505.4   128.2 1505.92   136.9 1507.18   144.3 1507.99
#Mann= 4 ,-1,0
       0      .1       0   66.62     .06       0    85.3    .045       0
    97.6     .06       0
Bank Sta=85.3,97.6
XS Rating Curve= 0 ,0
Exp/Cntr(USF)=0,0
Exp/Cntr=0.3,0.1

Type RM Length L Ch R = 1 ,3293    ,93.7,94.1,92
XS GIS Cut Line= 6
2152366.66364828648719.3111649722152343.38558717648716.168917219
2152332.76100311648715.8261887012152320.09065075 648731.07817743
2152290.76832197648775.6328847942152289.24508411648811.809783936
#Sta/Elev= 30
       0 1505.12     6.6 1504.22    18.7 1502.09    29.5 1499.74    34.1 1498.46
    35.9 1498.36    41.1 1497.35    49.7 1494.95    55.4 1494.07    58.3 1493.95
    64.1 1494.11    70.8 1495.01    75.6 1495.06    80.4 1494.03    85.2 1493.78
    87.2 1493.35    90.2 1492.51    92.9 1492.07    94.8 1492.05    97.5 1493.44
    99.6 1494.88   104.3 1499.05   107.3 1500.98   108.8 1501.85   112.8 1503.18
   116.8 1504.11   120.8 1504.74   128.9 1506.71   136.9 1507.02   143.5 1507.92
#Mann= 4 ,-1,0
       0      .1       0    87.2    .045       0    97.5      .1       0
  117.29     .06       0
Bank Sta=87.2,97.5
XS Rating Curve= 0 ,0
Exp/Cntr(USF)=0,0
Exp/Cntr=0.3,0.1

Type RM Length L Ch R = 1 ,3199    ,97.1,97.2,94.7
XS GIS Cut Line= 5
2152305.74031907648643.4007939142152263.89829147648653.273631886
2152219.70558816648722.8536328342152210.77302047648739.308362788
2152213.59383132648767.516471281
#Sta/Elev= 30
       0  1492.5     5.7 1492.55    13.9 1492.02      18 1491.53    26.3 1489.99
    34.5 1487.54      43 1485.88    47.6 1484.08    52.4 1482.66    57.1 1480.97
    60.1 1479.07    61.8 1478.24      63 1477.86    65.9 1477.32      76 1476.03
    80.8 1474.94    87.91472.763    90.3 1472.04      95 1471.88    99.7 1472.01
   102.2 1472.76   104.5  1473.9   109.2 1476.96   112.3 1478.34     114 1479.04
   123.9 1482.27   128.1 1484.04   138.6 1489.02   141.5 1490.14   172.5 1495.26
#Mann= 3 ,-1,0
       0      .1       0    87.9    .045       0   102.2      .1       0
Bank Sta=87.9,102.2
XS Rating Curve= 0 ,0
Exp/Cntr(USF)=0,0
Exp/Cntr=0.3,0.1

Type RM Length L Ch R = 1 ,3102    ,111.9,113.6,112.9
XS GIS Cut Line= 4
2152196.68397657648606.1018383432152165.79609777648633.181622496
2152131.10012433 648695.803623352152134.06197572648727.960867031
#Sta/Elev= 30
       0 1475.13     5.4 1474.38    11.3 1474.18    16.6 1474.19    22.4 1474.88
    25.2 1475.02    28.1 1474.71    30.9 1473.31    33.7 1471.63    36.6 1469.78
    41.1 1466.57    44.4 1465.06    45.6 1464.64    52.7 1463.64    59.4 1462.43
    71.7 1458.86    77.6 1458.09    83.5 1458.86    91.4 1460.29    95.9 1461.31
   105.1 1463.82   109.7 1464.15   112.7 1464.14   117.4 1464.73   122.1 1465.66
   126.1 1466.72   134.1 1469.64   138.2 1472.04   142.2 1474.85     145  1476.1
#Mann= 4 ,-1,0
       0      .1       0    71.7    .045       0    83.5      .1       0
  101.08     .06       0
Bank Sta=71.7,83.5
XS Rating Curve= 0 ,0
Exp/Cntr(USF)=0,0
Exp/Cntr=0.3,0.1

Type RM Length L Ch R = 1 ,2988    ,70.4,63.2,58.3
XS GIS Cut Line= 4
2152087.09547508648582.830148837 2152068.9012451648602.716865324
2152039.11034829648655.7272143952152044.36019071 648703.84293427
#Sta/Elev= 30
       0 1460.78     3.7 1459.32     6.6 1457.96     9.4 1456.29    16.2 1451.76
    19.4 1450.06    26.4 1447.55    29.8 1446.09    32.2 1445.19    35.2 1444.46
    36.6  1444.3    38.1 1443.95      39 1443.84      41 1443.16      44 1442.42
    46.9 1442.12    49.9 1442.18    53.81442.413    61.9 1443.35    82.2  1446.1
    87.8 1446.62      90 1447.04    93.2  1447.9    97.3  1449.2   111.8  1456.1
   113.4  1456.8   121.4 1459.93   125.4 1461.96   128.8 1463.84   136.2 1467.56
#Mann= 4 ,-1,0
       0      .1       0      10     .06       0      44    .045       0
    53.8     .06       0
Bank Sta=44,53.8
XS Rating Curve= 0 ,0
Exp/Cntr(USF)=0,0
Exp/Cntr=0.3,0.1

Type RM Length L Ch R = 1 ,2925    ,50.5,54.3,56
XS GIS Cut Line= 4
2152003.94692681648553.0673770222152000.65598082648576.574134099
2152000.65598082648630.169540235 2151999.2455754648695.518324909
#Sta/Elev= 30
       0 1444.03     8.2  1438.8    16.3 1434.36    20.3 1433.04    24.8 1433.09
    28.3 1433.65    31.9  1433.3    39.9 1430.08    44.3 1429.54    48.3 1429.48
    52.3 1429.67    56.3 1430.29    60.3 1431.75    68.3 1435.31    72.3 1435.75
    76.3 1435.87    80.3 1436.57    84.3 1438.13    88.3 1440.01    92.3 1441.29
    96.3 1441.92   104.3 1442.23   108.3    1443   112.3  1445.2   116.3 1447.86
   120.4 1449.65   124.4 1451.64   127.7 1453.66   136.4 1457.72   142.7 1461.95
#Mann= 5 ,-1,0
       0      .1       0   33.74     .06       0    39.9    .045       0
    56.3     .06       0  137.33      .1       0
Bank Sta=39.9,56.3
XS Rating Curve= 0 ,0
Exp/Cntr(USF)=0,0
Exp/Cntr=0.3,0.1

Type RM Length L Ch R = 1 ,2871    ,87.6,87.1,87.3
XS GIS Cut Line= 4
2151962.10489921648538.4931876342151958.81395322648548.366025607
2151940.94881785 648631.579945662151945.65016926648673.892108398
#Sta/Elev= 30
       0  1444.4     2.8 1444.42       7 1444.03    11.2 1442.47    13.3 1441.18
    15.3 1439.87    16.7 1438.51    19.4 1435.63    23.5 1430.47    27.6  1427.3
    31.7 1425.91    35.8 1424.91      44 1423.82    52.1 1422.07    56.2 1421.68
    60.3 1421.62      631422.082    68.5 1423.32    73.9 1425.66    77.3 1426.79
    80.8 1427.66    84.9 1428.08    93.1 1428.43   101.2 1428.53   105.2 1428.82
   109.2 1428.66   113.2 1429.36   121.3 1434.48   125.3 1436.71   138.1 1444.78
#Mann= 4 ,-1,0
       0      .1       0   50.41     .06       0    52.1    .045       0
      63     .06       0
Bank Sta=52.1,63
XS Rating Curve= 0 ,0
Exp/Cntr(USF)=0,0
Exp/Cntr=0.3,0.1

Type RM Length L Ch R = 1 ,2784    ,99.3,106.2,119.2
XS GIS Cut Line= 4
2151884.80695812648531.4775736822151872.53643092648542.478735994
2151857.72717397648611.8706828862151850.95722793648652.067237488
#Sta/Elev= 30
       0 1425.49     8.5 1419.35      13 1416.53    14.5 1415.72    15.8  1415.2
    19.1 1414.72    23.3  1414.3    27.4 1413.56    31.5 1412.61    35.6 1411.86
    39.7 1411.57    43.8 1411.41    47.9 1411.07      52 1410.64    56.1 1410.48
    59.5 1411.02    60.1 1411.14    64.2 1412.86    68.3 1414.78    72.4 1416.47
    76.5 1417.64    79.7  1418.2    84.7 1418.87    88.8 1419.78    92.8 1421.04
   100.9 1423.19     109 1425.53   113.1 1426.35   117.7 1427.95   128.2 1432.86
#Mann= 4 ,-1,0
       0      .1       0    47.9    .045       0    59.5      .1       0
   66.48     .06       0
Bank Sta=47.9,59.5
XS Rating Curve= 0 ,0
Exp/Cntr(USF)=0,0
Exp/Cntr=0.3,0.1

Type RM Length L Ch R = 1 ,2678    ,64.9,61.5,55.8
XS GIS Cut Line= 4
2151862.15203345648510.7773187462151851.80347118648515.822073468
 2151805.6832138648531.9006953092151785.79649731648546.709952268
#Sta/Elev= 26
       0 1422.62     2.2 1420.74     6.6 1416.78    11.1 1413.23    12.3 1412.56
    15.4 1411.09    19.6  1409.4    23.8 1406.42    28.1 1404.37    32.3 1403.86
    37.4 1404.09    39.9 1404.39    40.8 1404.51      45 1404.68    53.5 1404.56
    56.3 1404.81    60.4 1405.33    65.2 1406.22    67.2 1406.73    68.1 1407.01
    69.2  1407.5    70.9 1408.45    73.8 1410.31    77.2 1412.82    82.6 1416.67
    85.2  1418.4
#Mann= 4 ,-1,0
       0      .1       0    28.1    .045       0    39.9      .1       0
   60.36     .06       0
Bank Sta=28.1,39.9
XS Rating Curve= 0 ,0
Exp/Cntr(USF)=0,0
Exp/Cntr=0.3,0.1

Type RM Length L Ch R = 1 ,2616    ,44.1,48.8,53.7
XS GIS Cut Line= 2
2151816.34636699648463.5836017922151748.60950266648524.657823732
#Sta/Elev= 30
       0 1416.57     4.1 1413.79     5.6 1412.69     8.4 1410.24     9.7 1408.88
    14.3 1404.97    23.9  1398.3    26.3 1397.05    26.7 1396.89    27.2 1396.84
    29.6 1396.85    32.2 1397.09    35.3 1396.73    38.2 1396.58    40.9 1395.95
    44.2 1395.38    46.6  1395.2    49.4 1395.31    52.2    1396    54.1 1396.45
    59.5 1398.51    63.6 1400.66    68.1 1403.22    72.1 1405.76    74.1 1407.13
    77.7 1409.87      81  1412.2      86 1415.26      89 1417.25    91.2 1418.44
#Mann= 4 ,-1,0
       0      .1       0      40     .06       0    40.9    .045       0
    52.2     .06       0
Bank Sta=40.9,52.2
XS Rating Curve= 0 ,0
Exp/Cntr(USF)=0,0
Exp/Cntr=0.3,0.1

Type RM Length L Ch R = 1 ,2567    ,47.5,42.8,36.6
XS GIS Cut Line= 4
2151819.29603248648442.440552569 2151798.7528851648442.162942469
2151733.79212176648459.6523787522151724.07576827648476.864204935
#Sta/Elev= 30
       0 1422.54     3.1 1422.16     7.1  1420.5      10 1418.59    11.1 1417.81
    15.1 1414.57    19.1  1411.2    23.2 1407.45    27.4 1403.87    32.1 1400.35
    43.9 1391.86    48.1  1390.8    52.2 1390.81    56.4 1390.26    59.6 1390.04
    64.6 1389.58    68.8 1389.65    69.6 1389.99    77.1 1393.22    81.2  1394.3
    85.4 1394.63    87.1 1395.33    89.6 1396.98    90.1 1397.18    91.1 1397.52
    93.1 1397.84    98.8  1399.3   103.4 1401.71   104.8 1402.64   107.6 1404.28
#Mann= 3 ,-1,0
       0      .1       0    59.6    .045       0    69.6      .1       0
Bank Sta=59.6,69.6
XS Rating Curve= 0 ,0
Exp/Cntr(USF)=0,0
Exp/Cntr=0.3,0.1

Type RM Length L Ch R = 1 ,2524    ,85.2,100.6,84
XS GIS Cut Line= 2
2151851.67835616648318.9718268142151703.71154288648459.109503435
#Sta/Elev= 30
       0 1407.01       9 1400.65    15.8 1396.72    26.5 1388.58    29.5 1387.85
    40.8 1387.54    49.3 1387.91    60.6 1386.94    65.4 1387.22    76.4 1388.78
    83.3 1389.24    86.1 1389.63    91.8 1391.19    96.3 1391.54   100.2 1390.51
   105.9  1387.7   108.7 1386.69     120 1385.89   131.5 1386.44     137 1385.63
   142.6 1386.39   148.6 1389.62   153.6 1390.91   159.1 1391.22   164.6    1391
   170.1 1390.31   182.3 1390.39   186.6 1390.74   195.2 1392.44   203.8 1396.06
#Mann= 4 ,-1,0
       0      .1       0   131.5    .045       0   142.6      .1       0
     200     .06       0
#XS Ineff= 2 , 0
           95.41 1397.27
Permanent Ineff=
       F       F
Bank Sta=131.5,142.6
XS Rating Curve= 0 ,0
Exp/Cntr(USF)=0,0
Exp/Cntr=0.3,0.1

Type RM Length L Ch R = 1 ,2424    ,45.2,32.1,54.5
XS GIS Cut Line= 3
2151759.67822757648276.8930886362151692.72647352648362.659560348
2151644.81376504648421.959032655
#Sta/Elev= 30
       0 1401.89     5.7 1400.83    12.2  1397.2    18.7    1393    25.7 1387.54
    38.2 1377.14    44.7 1370.69      46 1370.03    51.1 1369.42      54 1370.45
    57.7 1371.76    62.5 1374.05    76.5 1377.73    85.3 1381.34    90.2 1381.55
    96.7 1379.94   103.2 1377.56   106.9 1377.16     112 1377.56   116.7 1378.73
   125.2 1380.13   136.6 1380.43   139.4 1381.31   142.9 1383.34     148 1385.35
   150.8 1385.88   160.6 1389.51     167 1391.38   178.9 1393.43     185 1393.29
#Mann= 4 ,-1,0
       0      .1       0    44.7    .045       0      54      .1       0
   148.8     .06       0
Bank Sta=44.7,54
XS Rating Curve= 0 ,0
Exp/Cntr(USF)=0,0
Exp/Cntr=0.3,0.1

Type RM Length L Ch R = 1 ,2392    ,87.7,93.6,75.3
XS GIS Cut Line= 4
2151747.58039466648263.6853013662151731.35489759648273.086470698
2151689.56510723648313.3091439192151607.10558148 648352.70852465
#Sta/Elev= 30
       0 1396.79     3.6 1395.29     8.6 1392.23    13.2 1387.95    17.8 1382.22
    21.1 1378.77    28.7    1370    30.4 1368.49    32.4 1367.35    35.2 1366.27
    39.8 1366.11    47.7 1366.39    53.5  1367.5      65 1372.29    67.6 1372.88
    73.1 1373.11    78.3 1372.54      96 1366.34   104.9 1365.03   109.3 1365.68
   118.2 1370.47   122.6 1371.11   131.5 1370.61   134.7 1370.92   144.8 1374.92
   149.7 1375.32   153.7 1375.19   158.1 1374.23   162.5 1372.71   168.1 1372.82
#Mann= 3 ,-1,0
       0      .1       0    32.4    .045       0    53.5      .1       0
#XS Ineff= 2 , 0
                           74.64         1378.18
Permanent Ineff=
       F       F
Bank Sta=32.4,53.5
XS Rating Curve= 0 ,0
Exp/Cntr(USF)=0,0
Exp/Cntr=0.3,0.1

Type RM Length L Ch R = 1 ,2298    ,93,89.4,80.6
XS GIS Cut Line= 4
2151660.59218849 648213.994357542151646.85048855648231.233944733
2151622.11542866 648274.957535442151617.61814505648307.937615288
#Sta/Elev= 30
       0 1389.19     2.6 1386.64     5.4 1384.19     7.1 1382.91     8.3 1382.12
    13.5 1378.92    14.3 1378.34    19.9 1373.67    22.5 1371.03    24.3 1369.43
    27.5 1365.72    31.3 1361.11    34.2 1357.96    35.6  1356.9    37.2 1355.92
    38.1 1355.55    40.1 1355.33    42.7 1355.16    47.3  1355.1    51.9 1355.38
    54.8  1356.2    56.5 1356.92      61 1359.76    65.6 1362.18    68.1 1363.16
    70.2 1363.86    74.5 1364.68    82.6 1365.83    98.7 1367.03   105.6 1367.46
#Mann= 3 ,-1,0
       0      .1       0    40.1    .045       0    51.9      .1       0
Bank Sta=40.1,51.9
XS Rating Curve= 0 ,0
Exp/Cntr(USF)=0,0
Exp/Cntr=0.3,0.1

Type RM Length L Ch R = 1 ,2209    ,55.9,65.1,71.8
XS GIS Cut Line= 5
2151552.02670919648199.9138708862151552.25157338648214.530042637
2151555.84940027648270.7460878322151557.19858535648291.433592463
2151556.74885699648299.978431333
#Sta/Elev= 26
       0 1358.76     1.3 1357.86     5.3 1355.77     9.3 1354.34    13.3 1353.25
    17.3 1351.49    21.3 1348.68    25.3 1346.63    29.3 1345.15    33.3 1344.35
    37.3    1344    41.3 1343.82    49.3 1344.01    53.3 1344.58    57.4 1346.14
    61.4 1348.15    64.6 1350.73      66 1351.67    69.4 1353.69    73.4 1354.95
    77.4 1355.79    81.4  1356.5    85.4 1358.02    93.4 1362.21    97.4 1363.77
   100.2 1365.17
#Mann= 3 ,-1,0
       0      .1       0    37.3    .045       0    49.3      .1       0
Bank Sta=37.3,49.3
XS Rating Curve= 0 ,0
Exp/Cntr(USF)=0,0
Exp/Cntr=0.3,0.1

Type RM Length L Ch R = 1 ,2144    ,54.7,62.3,56.1
XS GIS Cut Line= 4
2151533.17449843648192.3198173712151521.63896596648221.259837437
2151473.27068067648265.7829452312151467.60410331648284.604077162
#Sta/Elev= 30
       0 1365.43      .9 1364.86     2.7 1363.43     5.2 1361.25     9.5    1358
    13.8 1355.38    22.5 1350.62    26.8 1348.77      35  1346.4    36.9 1345.69
    38.6 1345.28    42.8 1343.83    46.3 1342.28    51.9 1339.98    54.9 1338.97
    59.91337.024    60.4 1336.85    63.3 1336.62    65.8  1336.7    68.9 1336.98
    72.4 1337.02    78.3 1337.39    85.9 1338.68    88.8 1339.43    91.6 1340.48
    94.4 1341.69    96.9 1342.64   100.4 1344.34     113 1351.22   116.6 1353.72
#Mann= 3 ,-1,0
       0      .1       0    59.9    .045       0    68.9      .1       0
Bank Sta=59.9,68.9
XS Rating Curve= 0 ,0
Exp/Cntr(USF)=0,0
Exp/Cntr=0.3,0.1

Type RM Length L Ch R = 1 ,2081    ,47.1,45.9,40.6
XS GIS Cut Line= 4
2151501.80594521648177.9509962192151478.93725803648184.427084626
2151442.91401626648243.5213913342151438.46170549648273.270922451
#Sta/Elev= 30
       0  1356.8     5.9 1353.53      10 1350.72    14.2 1347.75    22.5 1341.43
    26.3 1338.76      34 1333.03    35.1 1332.35    36.8 1331.37    38.7 1330.49
    44.4 1329.26    46.7 1329.03    52.5 1328.78    62.1 1328.97    64.2 1329.21
    67.1 1329.76      70 1331.28    71.5 1332.19    75.2 1334.83    76.2 1335.38
    81.6 1336.15    87.4 1337.36    90.2 1337.82    98.7 1337.87   102.7 1338.17
   103.9 1338.55   106.8 1339.56   110.9 1341.79   118.9 1346.53   123.1  1349.2
#Mann= 3 ,-1,0
       0      .1       0    46.7    .045       0    62.1      .1       0
Bank Sta=46.7,62.1
XS Rating Curve= 0 ,0
Exp/Cntr(USF)=0,0
Exp/Cntr=0.3,0.1

Type RM Length L Ch R = 1 ,2035    ,70.9,71.7,62.5
XS GIS Cut Line= 3
2151436.42052982648148.7553406632151416.63248191648227.457803936
2151412.80979083648258.713925064
#Sta/Elev= 30
       0 1342.14      .4 1341.78     4.6 1338.72     8.7 1335.22    12.8  1330.9
    13.7 1330.23    16.9 1328.22    21.1 1327.25    25.2 1326.96    29.3 1326.95
    33.8 1326.13    37.6 1325.52    41.7 1325.22    48.11326.159    54.1 1326.92
    58.2 1328.12    63.2 1330.07    66.6 1331.89    70.6 1333.19    78.8 1333.74
    82.9 1334.79    86.9 1336.27    90.9 1337.13      95 1337.17      99 1337.41
     103 1338.59   104.7 1339.41   107.1 1340.72   111.1 1343.21   112.6 1344.05
#Mann= 3 ,-1,0
       0      .1       0    33.8    .045       0    48.1      .1       0
Bank Sta=33.8,48.1
XS Rating Curve= 0 ,0
Exp/Cntr(USF)=0,0
Exp/Cntr=0.3,0.1

Type RM Length L Ch R = 1 ,1964    ,47.7,63.7,70
XS GIS Cut Line= 4
2151362.36525961648156.803257455 2151362.6151087648170.794806481
2151370.86012867648210.2709626622151369.86073231648249.497269753
#Sta/Elev= 27
       0 1335.55      .4 1335.38     4.4  1332.6     8.4 1328.53    12.4 1324.79
      14 1323.58    15.1 1322.87    16.4 1321.83    20.5 1319.42    22.81318.992
    24.6 1318.68    32.8 1318.61    36.9 1318.65    40.9 1318.99    40.9    1319
    44.4 1320.14    49.1 1322.27    53.2 1323.56    57.2 1324.43    65.2 1325.24
    69.2 1326.53    73.2 1328.94    77.2 1331.78    81.2 1334.02    85.2 1336.43
    89.2 1339.03    93.6    1342
#Mann= 3 ,-1,0
       0      .1       0    22.8    .045       0    40.9      .1       0
Bank Sta=22.8,40.9
XS Rating Curve= 0 ,0
Exp/Cntr(USF)=0,0
Exp/Cntr=0.3,0.1

Type RM Length L Ch R = 1 ,1900    ,51.9,61.6,69.2
XS GIS Cut Line= 4
2151341.87763425648165.7978246862151324.88789615648195.280017277
2151303.65072352 648222.013869882151297.15464719648249.747118843
#Sta/Elev= 30
       0 1323.28     3.9  1320.3     8.5 1318.05    13.1 1317.46    17.8 1316.97
    19.4 1316.91    22.4 1317.08    27.4 1317.87    30.1 1317.92    31.6 1318.11
      33 1318.06    35.2 1318.18    36.5 1317.98    38.7 1317.07    41.6 1316.12
    44.4 1314.94    46.7  1314.3      48 1314.09    50.1 1313.53    51.8 1313.36
    54.5 1313.47    58.91314.414    60.9 1314.81      62 1315.31    67.1 1319.26
    71.4 1323.75    79.6 1333.43    83.7 1336.79    87.9 1339.44    96.7 1344.61
#Mann= 3 ,-1,0
       0      .1       0    46.7    .045       0    58.9      .1       0
Bank Sta=46.7,58.9
XS Rating Curve= 0 ,0
Exp/Cntr(USF)=0,0
Exp/Cntr=0.3,0.1

Type RM Length L Ch R = 1 ,1838    ,112,101.2,84.9
XS GIS Cut Line= 5
2151355.69790233648142.6146657172151332.22208185648148.888376361
2151287.09184077648152.7335538532151256.56749986648157.225007656
2151249.92512301648171.025838543
#Sta/Elev= 28
       0 1336.98     7.8 1331.91    16.1 1327.86    20.2 1325.55    24.3 1323.12
    28.4 1320.52    32.4 1316.83    36.4 1311.73    37.2 1310.93    39.4 1308.53
    40.4 1307.56    43.1 1307.04    44.4 1306.82    48.4 1306.74    52.4 1307.14
    60.5 1308.59    64.5 1309.57    68.5 1310.24    72.6 1310.46    80.6 1309.94
    84.7  1309.5    88.7 1309.25    92.8  1309.6    97.2 1310.73   100.4  1311.9
   104.8 1314.19   109.3 1316.42   115.8 1319.28
#Mann= 3 ,-1,0
       0      .1       0    43.1    .045       0    52.4      .1       0
Bank Sta=43.1,52.4
XS Rating Curve= 0 ,0
Exp/Cntr(USF)=0,0
Exp/Cntr=0.3,0.1

Type RM Length L Ch R = 1 ,1737    ,52.7,53.1,52.5
XS GIS Cut Line= 4
2151248.84882865648059.6294805912151249.12643875648089.333761262
2151238.85486506648146.2438317062151239.96530546648167.619809384
#Sta/Elev= 30
       0 1333.48     1.5 1332.65     4.8 1330.47     8.8 1327.62    10.3 1326.41
    12.8  1324.6    17.6 1320.34    21.6 1316.28    24.6 1313.39    26.5 1311.97
    28.6 1310.23    29.6 1309.57    30.4  1309.2    33.6 1307.41    37.7 1306.01
    49.9 1302.25    53.9 1300.64    56.31299.776    57.9  1299.2    62.1 1298.64
    66.1 1298.82    68.51299.675    70.2  1300.4    74.3 1303.89    78.3 1307.49
      82 1309.94    85.5 1311.61    90.5 1313.65    99.2 1315.46   108.9 1317.93
#Mann= 3 ,-1,0
       0      .1       0    56.3    .045       0    68.5      .1       0
Bank Sta=56.3,68.5
XS Rating Curve= 0 ,0
Exp/Cntr(USF)=0,0
Exp/Cntr=0.3,0.1

Type RM Length L Ch R = 1 ,1684    ,103,99.3,96.5
XS GIS Cut Line= 4
 2151210.0925293648049.7421775012151199.34901844648073.977539207
2151188.85535667648136.4398116452151197.35022572  648161.9244188
#Sta/Elev= 29
       0 1325.83     4.7 1322.51    12.5 1318.39    13.2 1317.91    16.9 1314.77
    22.2 1309.76    25.6  1306.7    29.8 1304.12      32 1303.49    33.8 1303.07
    37.9 1302.32    41.9 1300.46      46  1298.8      50 1297.93    50.9 1297.86
    54.1 1297.61    58.1  1297.6    62.41298.086    66.3 1299.34    69.8 1300.81
    73.7  1302.3    78.4 1303.69    86.5 1305.71    90.6 1306.35    99.1 1307.33
   103.3 1307.35   107.5 1307.51   115.9 1308.38   116.7 1308.58
#Mann= 4 ,-1,0
       0      .1       0   46.51     .08       0    50.9    .045       0
    62.4     .08       0
Bank Sta=50.9,62.4
XS Rating Curve= 0 ,0
Exp/Cntr(USF)=0,0
Exp/Cntr=0.3,0.1

Type RM Length L Ch R = 1 ,1585    ,119.4,119.7,120.9
XS GIS Cut Line= 5
2151105.70210661 648028.054697682151104.45286117648054.538701194
2151113.69727749648125.2459935942151130.18731741648135.739655363
2151158.17041546648171.468075198
#Sta/Elev= 30
       0 1320.53     1.1 1319.68     5.1 1315.58     9.1 1311.66    13.1 1308.16
    21.1 1301.61    26.5 1297.96    33.2 1293.94    37.2 1292.08    39.3 1291.69
    41.3 1291.35    49.3 1291.38    53.1 1291.73    57.7 1292.09    61.4 1292.56
    65.5 1293.49    67.9  1293.8    73.6 1294.88    81.6 1293.62    85.7 1294.02
    93.7 1296.51    97.8 1296.49   105.4 1296.92   110.2 1297.49   127.1 1298.92
   129.4 1299.21   134.4 1300.58   139.5 1301.52   148.3 1302.12   162.8 1303.33
#Mann= 4 ,-1,0
       0      .1       0    39.3    .045       0    53.1      .1       0
   66.51     .08       0
Bank Sta=39.3,53.1
XS Rating Curve= 0 ,0
Exp/Cntr(USF)=0,0
Exp/Cntr=0.3,0.1

Type RM Length L Ch R = 1 ,1465    ,81.9,88.3,92
XS GIS Cut Line= 5
2151052.64169829648034.6831941582151018.91207117648068.662670364
 2151008.4184094648075.1587466982151005.17037123 648154.36090815
2150994.92655855648182.593855292
#Sta/Elev= 30
       0 1300.65     6.3 1297.59    14.8 1294.34    20.4 1292.62    26.1 1291.35
    33.2 1290.39      43 1289.89    48.9 1289.27    56.5  1287.8    70.2 1283.92
    78.3 1283.54    90.3 1282.25    94.3 1282.54    98.3  1283.3   102.3 1283.36
   106.3 1282.73   110.3 1282.53   114.3  1282.7   118.3 1283.31   122.3 1284.54
   126.3  1285.4   130.3 1285.84   134.3 1287.64   142.5 1293.35     151 1298.49
     155 1301.46   159.5  1305.5   164.3 1309.25     168 1311.55   169.5 1312.12
#Mann= 4 ,-1,0
       0      .1       0   80.22     .08       0   106.3    .045       0
   114.3     .08       0
Bank Sta=106.3,114.3
XS Rating Curve= 0 ,0
Exp/Cntr(USF)=0,0
Exp/Cntr=0.3,0.1

Type RM Length L Ch R = 1 ,1377    ,51.6,49.3,45.6
XS GIS Cut Line= 4
2150980.80213882648037.4092290312150963.13456014648057.262487551
2150940.36706183   648091.5048052150927.61726278648108.990243697
#Sta/Elev= 27
       0 1286.46       5 1285.46       7 1285.15    11.6 1284.15    17.3 1283.29
    20.1 1282.68      25 1281.45    28.7 1280.27    31.5 1279.23    37.3 1276.57
    39.1 1275.94    40.2 1275.64    40.9 1275.51    45.7 1275.29    48.8 1275.61
    55.3 1276.08    57.5 1276.36    60.1 1276.89    63.3 1278.09    64.9 1278.55
    67.7 1279.19    74.7 1280.71    77.6 1282.08    79.7 1283.17    81.6 1284.39
    84.6 1286.74    89.3 1290.97
#Mann= 4 ,-1,0
       0      .1       0    40.2    .045       0    48.8      .1       0
    67.7     .08       0
Bank Sta=40.2,48.8
XS Rating Curve= 0 ,0
Exp/Cntr(USF)=0,0
Exp/Cntr=0.3,0.1

Type RM Length L Ch R = 1 ,1328    ,71.3,69.6,64.7
XS GIS Cut Line= 5
2150928.76939542  648020.4609789 2150916.9302963648032.664357991
2150908.00543697648062.3531757792150907.45901701648082.024294313
2150906.54831708648108.981012305
#Sta/Elev= 30
       0 1285.43       1 1284.68     6.6 1281.28     9.4  1280.1    12.1 1279.37
    17.5 1276.95    19.6  1275.2    21.2 1273.66    21.7 1273.29    24.4 1272.17
    25.9 1271.73    30.1  1271.7    34.2 1271.98    34.71272.085    38.4  1272.9
    40.5 1273.48    42.6 1274.17    43.7  1274.6    46.5 1275.98    50.8  1277.7
    58.8 1279.91    62.3 1280.36    66.8 1281.14    70.8 1282.19    74.8 1283.64
    77.8 1285.07    81.7 1287.06    86.8 1290.12    90.9 1293.51    94.7 1298.22
#Mann= 4 ,-1,0
       0      .1       0    24.4    .045       0    34.7      .1       0
   77.68     .08       0
Bank Sta=24.4,34.7
XS Rating Curve= 0 ,0
Exp/Cntr(USF)=0,0
Exp/Cntr=0.3,0.1

Type RM Length L Ch R = 1 ,1258    ,53.9,53.5,51.8
XS GIS Cut Line= 4
2150855.55699435648021.0845192882150854.16894386648052.732070656
2150854.44655395648082.7139614272150864.44051754648111.030191598
#Sta/Elev= 21
       0  1280.4    14.8 1272.12    20.1  1269.5    24.1 1268.54    32.1  1268.5
    36.1  1268.1    40.41266.713    44.1 1265.52    48.1 1265.58      50 1266.64
    52.1 1267.84    56.1 1270.36    60.1 1272.43    61.8 1273.43    64.3 1275.08
    68.5  1278.3    74.4 1282.32    83.8 1289.29    85.5 1290.61    89.7 1294.51
    91.7 1295.97
#Mann= 4 ,-1,0
       0      .1       0    40.4    .045       0      50      .1       0
   71.66     .08       0
Bank Sta=40.4,50
XS Rating Curve= 0 ,0
Exp/Cntr(USF)=0,0
Exp/Cntr=0.3,0.1

Type RM Length L Ch R = 1 ,1204    ,51.4,49.7,44.4
XS GIS Cut Line= 4
2150800.03497441648029.6904323792150799.20214411648044.681377764
 2150805.3095663648092.1527048172150819.19007129648121.579375388
#Sta/Elev= 30
       0 1277.96     3.5 1275.08     3.8 1274.75     7.5  1271.6    11.5 1268.34
    15.5 1265.55    19.9 1263.25    23.5 1261.62      27  1260.2    27.6 1259.99
    30.6 1259.53    31.6 1259.35    35.7 1259.22    38.81259.551    43.7 1260.04
    47.8 1260.31    55.8 1261.48    59.9 1263.68    60.7 1264.54    62.9 1266.53
      64 1267.69    68.4 1271.67    69.6 1272.41    72.9 1274.15    77.3 1275.76
      79 1276.72    81.7 1278.53    83.8 1280.39    86.8 1282.82    95.4 1289.05
#Mann= 4 ,-1,0
       0      .1       0    30.6    .045       0    38.8      .1       0
   62.88     .08       0
Bank Sta=30.6,38.8
XS Rating Curve= 0 ,0
Exp/Cntr(USF)=0,0
Exp/Cntr=0.3,0.1

Type RM Length L Ch R = 1 ,1155    ,43.7,45.2,45.9
XS GIS Cut Line= 4
2150745.59804971648060.7637371652150752.88364917 648073.10878069
2150773.93093649648108.7272669252150796.59724591648133.214976211
#Sta/Elev= 27
       0 1264.67     2.2 1263.81     5.1 1263.03       8 1262.09    16.8 1259.95
    19.1 1259.23    20.8 1258.43    23.7  1256.9    25.6 1256.24    28.5  1255.5
      33 1255.36    37.2  1255.6    40.2 1256.15    43.1 1256.89      46 1257.93
    48.9 1259.29    51.8 1261.08    54.8  1262.7      59 1265.61    63.3 1268.33
    64.9 1269.47    68.9 1272.04    72.7 1274.71    78.1 1278.24    80.3 1279.36
    83.6 1281.17    89.1  1284.5
#Mann= 4 ,-1,0
       0      .1       0    25.6    .045       0    40.2      .1       0
   44.33     .08       0
Bank Sta=25.6,40.2
XS Rating Curve= 0 ,0
Exp/Cntr(USF)=0,0
Exp/Cntr=0.3,0.1

Type RM Length L Ch R = 1 ,1110    ,39.9,44.9,48.6
XS GIS Cut Line= 4
2150708.89976615648064.9523812212150712.36042589648088.084159498
 2150735.1279242648135.9869759292150748.24200322648162.761553934
#Sta/Elev= 29
       0 1263.28     4.3 1261.48     8.3 1259.11    12.4 1256.89    13.6 1256.38
    16.4 1255.41    20.7 1255.64    22.1 1255.88    24.6 1256.09      29 1254.35
    33.5 1252.14    36.1 1251.67    37.9 1251.44    42.3 1251.38    51.2 1251.54
    53.51251.714    55.6 1251.91    60.1 1252.66    64.5 1253.59    68.9 1255.25
    72.1 1256.78    77.8 1259.15    81.1 1260.78    86.7 1263.98    91.1  1266.7
    95.6 1269.85      99 1272.78     100 1273.56   106.2 1278.07
#Mann= 4 ,-1,0
       0      .1       0   33.39     .08       0    36.1    .045       0
    53.5     .08       0
Bank Sta=36.1,53.5
XS Rating Curve= 0 ,0
Exp/Cntr(USF)=0,0
Exp/Cntr=0.3,0.1

Type RM Length L Ch R = 1 ,1065    ,55.4,55.3,55
XS GIS Cut Line= 4
2150684.87020254648070.8860049842150682.37171164648087.625893997
2150681.37231528648142.5926937432150679.37352256648174.323528141
#Sta/Elev= 29
       0 1262.48     2.3 1261.89     6.7 1259.77    10.4 1257.59    13.2 1255.75
    16.2 1254.03    22.5 1250.16    26.5 1248.98    30.5 1248.53    34.5 1248.38
    38.5 1248.73    42.5 1248.53    46.5  1248.1    47.8 1247.85    50.5 1247.33
    54.5 1247.57    55.41247.874    62.5 1250.27    66.5 1252.18    67.8  1253.1
    69.2 1254.22    70.5 1255.12    78.5 1263.85    81.9 1267.19    82.5 1267.72
    86.5 1270.71    94.5 1275.54    98.5 1278.39   103.7 1282.51
#Mann= 4 ,-1,0
       0      .1       0   26.93     .08       0    47.8    .045       0
    55.4     .08       0
Bank Sta=47.8,55.4
XS Rating Curve= 0 ,0
Exp/Cntr(USF)=0,0
Exp/Cntr=0.3,0.1

Type RM Length L Ch R = 1 ,1009    ,79.9,89.8,94.5
XS GIS Cut Line= 3
 2150626.0381115648074.4426285742150627.27193417648151.865000831
2150625.11274451648177.466821139
#Sta/Elev= 23
       0 1253.53     6.7 1252.79    10.7 1251.74    22.7 1247.96    30.7 1246.36
    34.7 1245.44    42.7 1245.41      451245.117    46.7  1244.9    50.7 1244.65
    54.7 1245.12    58.7 1245.96    62.7  1248.2    65.7 1250.38    71.7 1255.27
    73.8  1256.8    78.8 1260.88    86.8 1269.39    90.8 1273.44    94.8 1278.01
     100 1283.02   101.8 1284.58   103.1 1285.83
#Mann= 5 ,-1,0
       0      .1       0      45    .045       0    54.7      .1       0
   77.43     .08       0   87.43      .1       0
Bank Sta=45,54.7
XS Rating Curve= 0 ,0
Exp/Cntr(USF)=0,0
Exp/Cntr=0.3,0.1

Type RM Length L Ch R = 1 ,920     ,63,61.7,58.7
XS GIS Cut Line= 4
2150619.86899818648061.4874905872150590.25725421 648065.49741425
2150551.39184025648103.745916879 2150533.5014116648124.103990859
#Sta/Elev= 30
       0 1254.39     7.8 1253.72    11.8 1253.14    15.8 1252.03    23.9 1248.77
    27.9 1247.87    29.9 1247.59      34 1246.48    38.4  1244.2      44 1240.46
    46.5 1239.42    49.6 1238.95    52.2 1238.78    55.3 1239.01    60.9 1239.98
    62.2 1240.05    65.1 1239.57    69.3 1237.71    70.61237.404    72.1 1237.04
      75  1237.4    80.8  1239.9      82 1240.22    89.3 1240.82    95.3 1242.04
    96.2 1242.53      99 1244.63   101.9 1247.33   108.8 1255.21   111.5 1258.58
#Mann= 3 ,-1,0
       0      .1       0    70.6    .045       0      75      .1       0
Bank Sta=70.6,75
XS Rating Curve= 0 ,0
Exp/Cntr(USF)=0,0
Exp/Cntr=0.3,0.1

Type RM Length L Ch R = 1 ,858     ,42.8,36.1,29
XS GIS Cut Line= 4
2150562.68818908648007.7107340012150550.19573459648026.449415732
2150528.70871287648050.684777438 2150515.7165602648084.164555465
#Sta/Elev= 30
       0 1252.18     8.6  1247.5    16.2  1243.5      19 1242.16    23.1 1240.04
    28.7 1236.95    31.6  1235.5    34.4 1234.36    36.9 1233.56    37.6 1233.43
    42.2 1233.05    43.7 1233.04    47.6 1233.13    49.7 1233.48    52.9 1234.67
    54.2 1234.98    56.4 1235.19    57.3 1235.13    60.3 1234.34    63.4 1233.14
    66.2 1231.71    67.4 1231.41    70.5 1231.17    74.7 1232.93    75.8  1233.3
    78.5 1234.75      79 1235.09    83.3 1236.27    88.2 1236.86    90.8 1237.35
#Mann= 3 ,-1,0
       0      .1       0    37.6    .045       0    49.7      .1       0
Bank Sta=37.6,49.7
XS Rating Curve= 0 ,0
Exp/Cntr(USF)=0,0
Exp/Cntr=0.3,0.1

Type RM Length L Ch R = 1 ,822     ,62.5,65.4,62.6
XS GIS Cut Line= 2
2150506.90350732647995.5952746232150499.22429864648081.602411742
#Sta/Elev= 24
       0 1240.13     1.6 1239.13     3.1 1238.33     9.6 1235.01    17.7 1230.74
    21.7 1228.98    25.7 1227.99    26.9  1227.9    29.7 1227.69    33.7 1227.64
    38.11227.849    41.7  1228.2    45.8 1228.98    49.8 1229.88    53.8 1231.26
    57.8 1232.34    61.8 1233.01    69.9 1235.94    73.9 1236.87    77.7 1238.01
    81.9 1238.45    85.1  1239.1    85.9 1239.34    86.3 1239.57
#Mann= 3 ,-1,0
       0      .1       0    26.9    .045       0    38.1      .1       0
Bank Sta=26.9,38.1
XS Rating Curve= 0 ,0
Exp/Cntr(USF)=0,0
Exp/Cntr=0.3,0.1

Type RM Length L Ch R = 1 ,756     ,41.4,40,40.4
XS GIS Cut Line= 4
2150450.25609869647992.2200904362150447.25790961648025.200170283
2150447.75760779648066.6751191822150451.75519323648097.406557222
#Sta/Elev= 29
       0  1235.6       1 1234.86       5 1232.19       9 1230.02    16.4 1226.69
      21 1224.24    25.1 1222.66    29.1 1222.12    33.1 1222.38    37.1 1222.11
    41.1 1220.92    45.1 1219.88    49.1 1219.47    53.1  1219.2    56.5 1219.98
    57.1  1220.1    61.1 1222.01    65.1 1223.01    69.1 1224.53    73.1 1226.93
    74.6 1227.95    77.8 1230.29    81.2 1232.61    81.6 1232.95    89.2 1237.94
    93.3 1240.39    97.3 1243.07   101.3 1246.31   105.6 1249.94
#Mann= 3 ,-1,0
       0      .1       0    45.1    .045       0    56.5      .1       0
Bank Sta=45.1,56.5
XS Rating Curve= 0 ,0
Exp/Cntr(USF)=0,0
Exp/Cntr=0.3,0.1

Type RM Length L Ch R = 1 ,716     ,69.6,70.1,70.3
XS GIS Cut Line= 4
2150413.95546557648012.902367572 2150409.9455419 648041.89720021
2150408.09480791 648081.687981172150404.08488424648109.757446809
#Sta/Elev= 25
       0 1224.45     4.3  1224.1     8.4 1222.96    16.4 1218.19    20.5 1217.12
    24.5 1217.27    28.5 1217.86    32.6 1217.63    36.6 1216.33    40.6 1215.79
    44.6 1216.06    45.41216.284    47.7 1217.17    48.6 1217.44    52.6 1219.37
    56.6  1221.9    64.5 1227.74    73.3 1234.94    76.7 1237.61    80.7  1241.3
    84.8 1244.66    89.8 1248.55    92.2 1250.26    92.8 1250.77    97.5 1253.39
#Mann= 3 ,-1,0
       0      .1       0    36.6    .045       0    45.4      .1       0
Bank Sta=36.6,45.4
XS Rating Curve= 0 ,0
Exp/Cntr(USF)=0,0
Exp/Cntr=0.3,0.1

Type RM Length L Ch R = 1 ,646     ,80.6,81.2,80
XS GIS Cut Line= 4
2150352.18396999647999.6312852482150344.30121407648016.424982639
 2150342.3270978648082.1089031482150356.55375859 648109.79108556
#Sta/Elev= 30
       0 1219.99     4.2 1217.93     6.1 1216.85    10.5 1214.73    13.2 1213.87
    16.2 1212.77    19.2 1211.98    31.6 1208.28    33.51207.888    35.3  1207.5
    39.3 1207.61    43.3 1207.88    47.3 1207.48    51.3 1207.47    59.3  1207.2
    63.3 1207.88    68.7 1209.44    75.3 1211.54    79.3 1212.19    81.1 1212.59
    83.3 1213.12    84.3 1213.61    87.9 1216.91    92.2 1220.04    96.7 1223.03
   105.7 1230.41   110.2 1234.49   114.6 1238.75   114.8 1239.06   115.4 1239.65
#Mann= 3 ,-1,0
       0      .1       0    33.5    .045       0    43.3      .1       0
Bank Sta=33.5,43.3
XS Rating Curve= 0 ,0
Exp/Cntr(USF)=0,0
Exp/Cntr=0.3,0.1

Type RM Length L Ch R = 1 ,565     ,87,89.5,89
XS GIS Cut Line= 4
2150267.17073243648005.7312842392150264.08617577648025.266809775
 2150266.4852754648107.8643826552150265.45708984648139.052677809
#Sta/Elev= 30
       0 1212.81     3.5 1212.27     7.5 1211.16    11.6 1209.11    15.6 1205.93
    19.7 1202.04    23.7 1199.06    27.7 1197.03    31.7 1195.69    35.7 1194.84
    39.7 1194.38    43.7 1194.22    48.4 1194.78    51.7  1195.1    60.8 1194.21
    63.7 1194.21    67.7 1194.97    75.7 1195.48    79.7 1196.11    83.7 1197.38
    87.7 1199.63    91.7 1202.09    95.7 1203.95   103.7 1209.08   111.7 1213.83
   115.7 1216.93   119.7 1220.24   123.7 1223.22   127.7 1225.75   133.6 1229.18
#Mann= 3 ,-1,0
       0      .1       0    35.7    .045       0    48.4      .1       0
Bank Sta=35.7,48.4
XS Rating Curve= 0 ,0
Exp/Cntr(USF)=0,0
Exp/Cntr=0.3,0.1

Type RM Length L Ch R = 1 ,476     ,75.9,80.3,76.3
XS GIS Cut Line= 4
2150215.55282083647987.6617036272150194.39673946648028.563460941
2150191.10579347 648101.904543022150191.10579347648139.515354342
#Sta/Elev= 30
       0 1211.71    10.7 1207.73    15.5 1205.24    24.2 1201.55    28.7 1199.27
    33.2 1196.34    37.7 1195.43    46.7 1194.79    50.7 1194.22    54.7 1193.05
    64.1 1189.02    70.7 1186.89    74.7 1186.42    77.31186.895    82.7 1188.21
    86.7 1188.99    94.7  1189.1    98.6 1190.23   102.4 1192.05   106.7 1194.87
   110.7 1197.11   114.7 1198.74   118.7 1201.02   122.7 1204.14   127.8 1207.74
   134.7 1213.14   138.7 1215.95   145.7 1220.42   154.7 1227.03   157.1 1228.36
#Mann= 4 ,-1,0
       0      .1       0    70.7    .045       0    77.3      .1       0
  116.05     .06       0
Bank Sta=70.7,77.3
XS Rating Curve= 0 ,0
Exp/Cntr(USF)=0,0
Exp/Cntr=0.3,0.1

Type RM Length L Ch R = 1 ,395     ,217.5,136.1,208.2
XS GIS Cut Line= 3
2150155.97888016647953.5723140532150133.87070772647982.833130511
 2150102.0089298648152.545865969
#Sta/Elev= 30
       0 1209.79     9.5 1206.36    14.5 1204.05    19.6 1200.87    25.3  1196.3
    33.8 1190.31    39.1 1187.52    43.1 1186.07    47.5 1185.43    71.6 1185.23
    75.7 1184.53    83.8 1181.81    87.9 1181.13    98.4  1182.2   104.2    1182
   120.5 1179.39   125.8 1178.04   128.6 1177.16   132.7 1176.56   136.7 1177.01
   139.5  1177.9   146.4 1180.63   154.3 1186.68   169.3 1200.75   177.4 1209.41
   185.6 1217.45   189.6 1220.13   193.7 1221.94   204.6 1225.73   209.4 1226.79
#Mann= 4 ,-1,0
       0      .1       0   125.8    .045       0   139.5      .1       0
  146.67     .06       0
Bank Sta=125.8,139.5
XS Rating Curve= 0 ,0
Exp/Cntr(USF)=0,0
Exp/Cntr=0.3,0.1

Type RM Length L Ch R = 1 ,259     ,168.4,168.4,168.4
XS GIS Cut Line= 3
  2149965.458453647905.4545269882149955.70484751 647950.97135259
2150034.38393176648159.048269626
#Sta/Elev= 30
       0 1196.29     7.9 1195.38    20.2 1191.32    28.4 1187.78    53.2 1173.73
    57.9 1171.93    67.2 1171.23    82.8 1171.38      96  1170.3   104.5 1171.47
   113.1 1170.57   126.2 1170.48   135.5 1172.24   149.7 1173.45   157.2 1175.06
     161 1175.46   181.5 1173.41   194.3 1170.48   197.6 1169.45   202.9 1168.87
   207.1 1169.48   211.4 1173.02   215.7 1178.35   228.3 1192.36   232.8 1196.79
   237.9 1199.95   240.1 1200.99   254.2 1206.16   262.7 1210.44     269 1213.14
#Mann= 3 ,-1,0
       0      .1       0   197.6    .045       0   207.1      .1       0
#XS Ineff= 2 , 0
          161.92 1180.44
Permanent Ineff=
       F       F
Bank Sta=197.6,207.1
XS Rating Curve= 0 ,0
Exp/Cntr(USF)=0,0
Exp/Cntr=0.3,0.1
